--- Hec-aguacatal.prj (project) ---

Proj Title=Hec-aguacatal
Current Plan=p01
Default Exp/Contr=0.3,0.1
SI Units
Geom File=g01
Flow File=f01
Plan File=p01
Y Axis Title=Elevation
X Axis Title(PF)=Main Channel Distance
X Axis Title(XS)=Station
BEGIN DESCRIPTION:
END DESCRIPTION:
DSS Export Rating Curves= 0
DSS Export Rating Curve Sorted= 0
DSS Export Volume Flow Curves= 0
DXF OffsetX= 0
DXF OffsetY= 0
DXF ScaleX= 1
DXF ScaleY= 10

--- Hec-aguacatal.p01 (plan) ---

Plan Title=Plan 01
Program Version=4.00
Short Identifier=Plan 01
Geom File=g01
Flow File=f01
Mixed Flow
K Sum by GR= 0
Std Step Tol= 0.003
Critical Tol= 0.003
Num of Std Step Trials= 20
Max Error Tol= 0.1
Flow Tol Ratio= 0.001
Split Flow NTrial= 30
Split Flow Tol= 0.006
Split Flow Ratio= 0.02
Log Output Level= 0
Friction Slope Method= 1
Unsteady Friction Slope Method= 2
Unsteady Bridges Friction Slope Method= 1
Parabolic Critical Depth
Global Vel Dist= 6 , 6 , 6
Global Log Level= 0
CheckData=True
Encroach Param=-1 ,0,0, 0
Computation Interval=1HOUR
Output Interval=1HOUR
Run HTab= 0
Run UNet= 0
Run PostProcess= 0
Run WQNet= 0
UNET Theta= 1
UNET Theta Warmup= 1
UNET ZTol= 0.006
UNET ZSATol= 0.015
UNET MxIter= 20
UNET MaxInSteps= 0
UNET DtIC= 0
UNET DtMin= 0
UNET MaxCRTS= 20
UNET WFStab= 2
UNET SFStab= 1
UNET WFX= 1
UNET SFX= 1
UNET DSS MLevel= 4
UNET DZMax Abort= 30
UNET Convert EG Bridges= 0
UNET Use Existing IB Tables=-1
UNET Froude Reduction=False
UNET Froude Limit= 1
UNET Froude Power= 10
UNET Time Slicing=0,0, 5
Instantaneous Interval=1HOUR
Write IC File= 0
Echo Input=False
Echo Output=False
Write Detailed= 0
Detailed Automatic Start=False, 10
WQ ULTIMATE=-1
WQ Max Comp Step=1HOUR
WQ Output Interval=15MIN
WQ Output Selected Increments= 0
WQ Output face flow=0
WQ Output face velocity=0
WQ Output face area=0
WQ Output face dispersion=0
WQ Output cell volume=0
WQ Output cell surface area=0
WQ Output cell continuity=0
WQ Output face conc=0
WQ Output face dconc_dx=0
WQ Output face courant=0
WQ Output face peclet=0
WQ Output face adv mass=0
WQ Output face disp mass=0
WQ Output cell mass=0
WQ Output cell source sink temp=0
WQ Output cell source sink nsm=0
WQ Output MaxMinRange=-1
WQ Daily Max Min Mean=-1
WQ Daily Range=0
WQ Daily Time=0
WQ Create Restart=0
WQ Fixed Restart=0
WQ System Summary=False
Sorting and Armoring Iterations= 10
XS Update Threshold= 0.02
Hydraulics Update Threshold= 0.02
Energy Slope Method= 1
Volume Change Method= 0
XS Weighting Method= 0
Number of US Weighted Cross Sections= 1
Number of DS Weighted Cross Sections= 1
Upstream XS Weight=0.25
Main XS Weight=0.5
Downstream XS Weight=0.25
Number of DS XS's Weighted with US Boundary= 1
Upstream Boundary Weight= 1
Weight of XSs Associated with US Boundary= 0
Number of US XS's Weighted with DS Boundary= 1
Downstream Boundary Weight= 0.5
Weight of XSs Associated with DS Boundary= 0.5
Sediment Output Level= 4
Mass or Volume Output= 0
Output Increment Type= 1
Profile and TS Output Increment= 10
XS Output Flag= 0
XS Output Increment= 10
Disregard all LS=0
Disregard all Conn=0
Disregard all Breaches=0
Disregard all Pumps=0

--- Hec-aguacatal.f01 (steady flow) ---

Flow Title=aguacatal
Program Version=4.00
Number of Profiles= 5
Profile Names=5 años,10 años,25 años,50 años,100 años
River Rch & RM=1,1               ,57
   31.09   41.67   55.03   64.95   74.79
Boundary for River Rch & Prof#=1,1               , 1
Up Type= 3
Up Slope=0.021398
Dn Type= 3
Dn Slope=0.013995
Boundary for River Rch & Prof#=1,1               , 2
Up Type= 3
Up Slope=0.021398
Dn Type= 3
Dn Slope=0.013995
Boundary for River Rch & Prof#=1,1               , 3
Up Type= 3
Up Slope=0.021398
Dn Type= 3
Dn Slope=0.013995
Boundary for River Rch & Prof#=1,1               , 4
Up Type= 3
Up Slope=0.021398
Dn Type= 3
Dn Slope=0.013995
Boundary for River Rch & Prof#=1,1               , 5
Up Type= 3
Up Slope=0.021398
Dn Type= 3
Dn Slope=0.013995
DSS Import GetInterval= 0
DSS Import GetPeak= 0
DSS Import FillOption= 0

--- Hec-aguacatal.g01 (geometry) ---

Geom Title=HEC-AGUACATAL
Program Version=4.00

River Reach=1               ,1
Reach XY= 4
1.267857142857140.293367346938780.920918367346940.47704081632653
0.31122448979592 0.4515306122449-0.29336734693870.83418367346939

Type RM Length L Ch R = 1 ,57      ,102,100.2,98.14
BEGIN DESCRIPTION:
S0
END DESCRIPTION:
#Sta/Elev= 24
       0 1133.04       1 1133.13    2.62 1133.11    3.75 1132.99     4.2 1132.75
    4.21 1132.87    5.58 1132.74    7.06 1131.91    7.77 1131.35   10.03 1130.43
   12.29 1131.13   13.13 1131.76   13.37 1132.17   13.76 1132.57    14.1 1132.65
   15.59 1132.65   16.82 1132.26   17.79 1132.65   18.03 1132.65   18.63 1133.06
   18.82 1133.45   19.63 1134.39   20.65 1134.06   24.65 1133.89
#Mann= 3 , 0 , 0
       0     .06       0    5.58    .045       0   13.76     .06       0
Levee=-1,1.45,1133.14,-1,19.59,1134.39,,
Bank Sta=5.58,13.76
XS Rating Curve= 0 ,0
Exp/Cntr=0.3,0.1

Type RM Length L Ch R = 1 ,56      ,110.44,110.1,109.85
BEGIN DESCRIPTION:
S100
END DESCRIPTION:
#Sta/Elev= 24
      .3 1130.64     2.8 1130.04     3.5 1130.04     3.5 1131.54    5.71 1131.54
    5.71 1128.04    8.71 1127.84   11.71 1128.04    11.8 1128.16    11.8 1128.21
   11.84 1128.34    11.9 1128.38   12.01 1128.64   12.01 1131.54   12.81 1131.54
   12.81 1128.94   13.14  1129.1   13.35 1129.26   13.54 1129.37   13.71 1129.46
   13.91 1129.63   14.07 1129.63   14.77 1130.34   14.77 1131.54
#Mann= 3 , 0 , 0
      .3     .06       0    5.71    .045       0   12.01     .06       0
Levee=-1,3.5,1131.56,-1,12.81,1131.54,,
Bank Sta=5.71,12.01
XS Rating Curve= 0 ,0
Exp/Cntr=0.3,0.1

Type RM Length L Ch R = 1 ,55      ,130.15,134.5,139.14
BEGIN DESCRIPTION:
S200
END DESCRIPTION:
#Sta/Elev= 23
       0 1133.17     .19 1131.03     .31 1132.04     .77 1130.36     1.5 1129.43
    1.94 1129.07    2.26 1128.63    2.44 1127.87    2.44 1128.19    2.68 1127.75
    2.91 1127.47     3.1 1127.38    3.32 1127.13     3.4 1126.89     3.5 1126.43
     5.5 1126.16     8.2 1125.93    10.9  1126.1    11.4 1126.33    13.4 1127.31
    14.4 1127.88    14.5 1128.11   14.65 1130.11
#Mann= 3 , 0 , 0
       0     .06       0     3.1    .045       0    13.4     .06       0
Levee=-1,0.01,1133.22,-1,14.67,1130.13,,
Bank Sta=3.1,13.4
XS Rating Curve= 0 ,0
Exp/Cntr=0.3,0.1

Type RM Length L Ch R = 1 ,54      ,119.63,123.5,126.4
BEGIN DESCRIPTION:
S300
END DESCRIPTION:
#Sta/Elev= 21
       01130.408    .1081129.947    .5421129.622   1.1931129.487   1.5731129.161
   1.8711128.592   2.5221128.538   2.849 1127.89   6.849 1127.51  12.849 1126.81
  13.349 1124.63  22.349  1124.7  32.349  1125.7  33.0931126.855  33.4861126.895
  33.6431127.837  34.0351128.425  34.7031128.975  34.8211129.485  34.8991129.642
  35.3321129.878
#Mann= 3 , 0 , 0
       0     .06       0  12.849    .045       0  33.093     .06       0
Levee=-1,0.06,1130.42,-1,35.34,1129.89,,
Bank Sta=12.849,33.093
XS Rating Curve= 0 ,0
Exp/Cntr=0.3,0.1

Type RM Length L Ch R = 1 ,53      ,161.62,132.02,105.11
BEGIN DESCRIPTION:
S400
END DESCRIPTION:
#Sta/Elev= 20
       0  1126.9      .4  1126.5      .6  1126.1     1.2  1125.7     2.2  1124.5
     3.2  1124.2     4.2  1123.6     5.2  1123.4     7.2  1122.8     9.9  1122.8
    12.7  1122.7    13.7    1125    14.7  1125.5    15.7  1126.3    16.7  1127.1
    17.5  1127.9    17.5  1128.6      18  1129.3    18.3    1130    18.3  1130.3
#Mann= 3 , 0 , 0
       0     .06       0     3.2    .045       0    13.7     .06       0
Levee=-1,0.02,1126.94,-1,18.3,1130.32,,
Bank Sta=3.2,13.7
XS Rating Curve= 0 ,0
Exp/Cntr=0.3,0.1

Type RM Length L Ch R = 1 ,52      ,124.4,1.22,119.8
BEGIN DESCRIPTION:
S500
END DESCRIPTION:
#Sta/Elev= 16
   -2.49 1119.53   -1.97  1119.1   -1.33 1118.85    -.67 1118.35       0 1117.48
     3.5 1117.37     5.5 1117.25     7.5 1116.98     8.5 1115.82      14  1115.9
      24 1116.95   24.68 1118.53   25.21 1118.84   25.39 1120.17   25.64 1120.91
   26.26 1122.06
#Mann= 3 , 0 , 0
   -2.49     .06       0     7.5    .045       0      24     .06       0
Levee=-1,-2.51,1119.53,-1,26.3,1122.06,,
Bank Sta=7.5,24
XS Rating Curve= 0 ,0
Exp/Cntr=0.3,0.1

Type RM Length L Ch R = 1 ,51      ,101.6,10,101.88
BEGIN DESCRIPTION:
S600
END DESCRIPTION:
#Sta/Elev= 23
   -3.34 1119.41   -2.91 1119.06   -2.05 1118.64   -1.17 1118.18    -.97 1118.14
    -.76  1118.1    -.02 1118.05     .38 1117.69     .64 1117.57    1.08 1116.92
    1.15 1116.61    1.75 1116.15       2 1115.51     2.8 1115.14     3.3 1114.12
       4 1113.36     4.5  1113.2       7 1113.13     9.5 1113.11    10.5 1118.86
   11.07 1119.32   11.24  1119.9   11.46 1120.35
#Mann= 3 , 0 , 0
   -3.34     .06       0     3.3    .045       0    10.5     .06       0
Levee=-1,-3.33,1119.41,-1,11.47,1120.35,,
Bank Sta=3.3,10.5
XS Rating Curve= 0 ,0
Exp/Cntr=0.3,0.1

Type RM Length L Ch R = 1 ,50      ,106.21,104.2,103.9
BEGIN DESCRIPTION:
S700
END DESCRIPTION:
#Sta/Elev= 17
     .44 1112.82      .7 1112.47    1.52 1112.48    2.52 1112.22    3.52 1111.59
    4.52 1110.67    7.72 1110.65   10.92 1110.81   11.92 1111.09   12.92 1111.49
   13.92 1112.07   14.92 1112.35   15.92 1112.48   16.81 1113.48   17.27 1113.98
   17.44 1114.73   17.66 1115.25
#Mann= 3 , 0 , 0
     .44     .06       0    3.52    .045       0   12.92     .06       0
Levee=-1,0.44,1112.82,-1,17.67,1115.26,,
Bank Sta=3.52,12.92
XS Rating Curve= 0 ,0
Exp/Cntr=0.3,0.1

Type RM Length L Ch R = 1 ,49      ,103.2,103.5,103.9
BEGIN DESCRIPTION:
S800
END DESCRIPTION:
#Sta/Elev= 9
       01106.983     1.2 1107.04     2.2 1106.56    4.45  1106.4     6.7 1106.68
     7.7 1107.19     8.7 1107.26     9.7 1107.49    10.7 1108.06
#Mann= 3 , 0 , 0
       0     .06       0     1.2    .045       0    10.7     .06       0
Levee=-1,1.19,1107.05,-1,10.69,1108.07,,
Bank Sta=1.2,10.7
XS Rating Curve= 0 ,0
Exp/Cntr=0.3,0.1

Type RM Length L Ch R = 1 ,48      ,100.06,110.5,127.06
BEGIN DESCRIPTION:
S900
END DESCRIPTION:
#Sta/Elev= 16
       0  1109.2      .6  1109.1     1.6    1108     2.9  1107.4     4.9  1104.2
     5.9  1103.9     8.9  1103.5    11.9  1103.2    12.1  1102.5    14.7  1102.7
    17.9    1103    18.9    1103    19.9  1103.3    20.8  1103.8    21.5  1104.9
    22.5  1105.8
#Mann= 3 , 0 , 0
       0     .06       0     5.9    .045       0    20.8     .06       0
Levee=-1,0.08,1109.25,-1,22.45,1105.82,,
Bank Sta=5.9,20.8
XS Rating Curve= 0 ,0
Exp/Cntr=0.3,0.1

Type RM Length L Ch R = 1 ,47      ,107.23,107.5,107.77
BEGIN DESCRIPTION:
S1000
END DESCRIPTION:
#Sta/Elev= 12
       0  1102.2     7.3 1102.06     8.3 1101.49    13.6 1100.48    16.9 1100.16
    17.4 1099.51   19.05 1099.25    20.7 1099.56    21.7 1100.54    22.7 1100.94
    23.7 1101.06    33.7 1101.03
#Mann= 3 , 0 , 0
       0     .06       0     8.3    .045       0    23.7     .06       0
Levee=-1,0.03,1102.21,-1,23.76,1101.05,,
Bank Sta=8.3,23.7
XS Rating Curve= 0 ,0
Exp/Cntr=0.3,0.1

Type RM Length L Ch R = 1 ,46      ,112.97,99.8,96.6
BEGIN DESCRIPTION:
S1100
END DESCRIPTION:
#Sta/Elev= 17
       01101.584     .39 1101.32     .78  1100.7    1.21 1100.68    1.56 1100.32
     2.5 1100.06     3.5 1099.89     4.5 1099.84     5.5 1099.56     6.5 1098.56
     8.3 1097.76    10.9 1097.68   14.86 1097.02   15.86 1098.71   17.46 1099.08
   19.46 1098.98   21.11 1099.14
#Mann= 3 , 0 , 0
       0     .06       0     5.5    .045       0   17.46     .06       0
Levee=-1,0.04,1101.6,-1,21.1,1099.17,,
Bank Sta=5.5,17.46
XS Rating Curve= 0 ,0
Exp/Cntr=0.3,0.1

Type RM Length L Ch R = 1 ,45      ,97.27,101.3,104.3
BEGIN DESCRIPTION:
S1200
END DESCRIPTION:
#Sta/Elev= 12
       0  1098.1     3.6  1097.6     5.6  1097.5     7.6  1097.3     8.6  1097.1
     9.6  1096.2    12.2  1096.1    14.9  1096.2    15.9  1096.7    17.9  1096.9
    19.9    1097    21.9  1096.8
#Mann= 3 , 0 , 0
       0     .06       0     7.6    .045       0    19.9     .06       0
Levee=-1,0.02,1098.11,-1,19.9,1096.99,,
Bank Sta=7.6,19.9
XS Rating Curve= 0 ,0
Exp/Cntr=0.3,0.1

Type RM Length L Ch R = 1 ,44      ,95.01,100,103.64
BEGIN DESCRIPTION:
S1300
END DESCRIPTION:
#Sta/Elev= 16
       0 1094.54     1.2 1094.33    2.15 1094.31    3.15 1094.34    4.15 1094.43
    5.25  1092.8    6.15 1092.03    8.65 1091.92   11.15 1092.11   12.15 1092.59
   13.35  1093.6   15.35 1093.64   17.35 1093.65   19.35 1093.65   21.35 1093.72
   26.35 1093.99
#Mann= 3 , 0 , 0
       0     .06       0    4.15    .045       0   13.35     .06       0
Levee=-1,0.09,1094.55,-1,26.34,1094.01,,
Bank Sta=4.15,13.35
XS Rating Curve= 0 ,0
Exp/Cntr=0.3,0.1

Type RM Length L Ch R = 1 ,43      ,95.42,99.2,102.4
BEGIN DESCRIPTION:
S1400
END DESCRIPTION:
#Sta/Elev= 17
       0  1092.3       5 1092.09      10  1091.6      15 1091.45      20  1091.5
      27  1091.3      28 1091.39      29 1091.42      30 1091.85      31 1093.25
      32 1096.05  33.4851096.262   34.041096.737  34.5121097.036  34.742 1097.45
    35.21097.633  35.2021097.634
#Mann= 3 , 0 , 0
       0     .06       0       0    .045       0      31     .06       0
Levee=-1,0.12,1092.33,-1,35.24,1097.61,,
Bank Sta=0,31
XS Rating Curve= 0 ,0
Exp/Cntr=0.3,0.1

Type RM Length L Ch R = 1 ,42      ,74.26,66.3,56.26
BEGIN DESCRIPTION:
S1500
END DESCRIPTION:
#Sta/Elev= 15
       0 1091.42       2 1091.37       4 1089.65       6 1088.97       8 1087.91
    10.5 1087.91      13 1088.02      15 1088.74      17 1089.56      19 1090.76
      21 1091.78      23 1092.97      28 1093.24      30 1092.89      32 1092.14
#Mann= 3 , 0 , 0
       0     .06       0       6    .045       0      15     .06       0
Levee=-1,0.08,1091.43,-1,27.97,1093.25,,
Bank Sta=6,15
XS Rating Curve= 0 ,0
Exp/Cntr=0.3,0.1

Type RM Length L Ch R = 1 ,41      ,99.05,100.6,102.15
BEGIN DESCRIPTION:
S1600
END DESCRIPTION:
#Sta/Elev= 10
       0 1087.83       5 1087.72      10 1087.39      15 1086.41   18.25 1086.46
    21.5  1086.3      24 1087.27      25 1089.06    25.5 1091.96  32.519 1091.96
#Mann= 3 , 0 , 0
       0     .06       0      10    .045       0      24     .06       0
Levee=-1,0.08,1087.88,-1,25.46,1091.97,,
Bank Sta=10,24
XS Rating Curve= 0 ,0
Exp/Cntr=0.3,0.1

Type RM Length L Ch R = 1 ,40      ,107.8,104.3,98.86
BEGIN DESCRIPTION:
S1700
END DESCRIPTION:
#Sta/Elev= 12
       0 1085.93     2.9 1085.93     5.9  1086.3     7.9  1084.8    10.9 1084.08
    11.4 1083.75      14  1083.6    16.6 1084.08    16.8 1084.14      20 1084.08
      25 1085.92      30 1086.38
#Mann= 3 , 0 , 0
       0     .06       0     7.9    .045       0      25     .06       0
Levee=-1,5.91,1086.3,-1,29.81,1086.37,,
Bank Sta=7.9,25
XS Rating Curve= 0 ,0
Exp/Cntr=0.3,0.1

Type RM Length L Ch R = 1 ,39      ,102.2,99.2,97.87
BEGIN DESCRIPTION:
S1800
END DESCRIPTION:
#Sta/Elev= 10
       01088.943       31088.943     8.61084.143     9.21082.982      101082.663
    12.3  1082.5    14.61082.803    16.61083.652    18.61084.563    21.41084.563
#Mann= 3 , 0 , 0
       0     .06       0     8.6    .045       0    18.6     .06       0
Levee=-1,2.99,1088.94,-1,18.57,1084.57,,
Bank Sta=8.6,18.6
XS Rating Curve= 0 ,0
Exp/Cntr=0.3,0.1

Type RM Length L Ch R = 1 ,38      ,103.41,102.5,101.32
BEGIN DESCRIPTION:
S1900
END DESCRIPTION:
#Sta/Elev= 11
       0  1083.7     5.3  1083.7     6.3    1083     7.3  1080.8     8.3    1080
    10.8  1079.3    13.3  1080.1    13.8  1080.2    15.8  1080.6    15.8  1084.1
    19.3  1084.1
#Mann= 3 , 0 , 0
       0     .06       0     7.3    .045       0    15.8     .06       0
Levee=-1,5.28,1083.71,-1,19.27,1084.12,,
Bank Sta=7.3,15.8
XS Rating Curve= 0 ,0
Exp/Cntr=0.3,0.1

Type RM Length L Ch R = 1 ,37      ,89.15,94.2,98.31
BEGIN DESCRIPTION:
S2000
END DESCRIPTION:
#Sta/Elev= 14
       0 1080.47       5 1080.47       6 1080.62       7 1079.52       8 1078.77
      14 1079.27      20 1078.97    21.5 1080.17    22.6 1081.94    23.6 1083.35
    24.6 1084.37    25.6 1085.14    26.6 1085.86    31.7 1085.86
#Mann= 3 , 0 , 0
       0     .06       0       7    .045       0    21.5     .06       0
Levee=-1,6.03,1080.62,-1,26.68,1085.89,,
Bank Sta=7,21.5
XS Rating Curve= 0 ,0
Exp/Cntr=0.3,0.1

Type RM Length L Ch R = 1 ,36      ,109.53,106.2,104.85
BEGIN DESCRIPTION:
S2100
END DESCRIPTION:
#Sta/Elev= 18
    -.151078.121       0 1078.13       0 1076.13       1 1076.13       3 1075.66
       5 1074.83       7 1074.49     7.5 1074.33    9.75 1074.08      12 1074.27
      14 1074.54      16  1074.4      17 1075.08  17.1751075.924   17.321077.326
  17.3781080.261    17.5 1083.15  22.803 1083.15
#Mann= 3 , 0 , 0
    -.15     .06       0       3    .045       0      17     .06       0
Levee=-1,0.03,1078.05,-1,17.52,1083.16,,
Bank Sta=3,17
XS Rating Curve= 0 ,0
Exp/Cntr=0.3,0.1

Type RM Length L Ch R = 1 ,35      ,97.37,99.2,101.7
BEGIN DESCRIPTION:
S2200
END DESCRIPTION:
#Sta/Elev= 18
       0  1086.6     5.8  1086.6     7.1  1087.3     8.4  1087.3    10.5  1086.2
    15.5  1073.1    17.5  1072.4    19.5  1072.1      22  1071.5    24.5  1071.4
    25.5  1073.6    26.1  1075.6    26.9  1077.1    27.5  1078.5    28.5  1080.1
    29.5  1081.4      31  1082.4    34.9  1082.4
#Mann= 3 , 0 , 0
       0     .06       0    15.5    .045       0    25.5     .06       0
Levee=-1,8.41,1087.29,-1,31.05,1082.42,,
Bank Sta=15.5,25.5
XS Rating Curve= 0 ,0
Exp/Cntr=0.3,0.1

Type RM Length L Ch R = 1 ,34      ,98.92,98.05,97.7
BEGIN DESCRIPTION:
S2300
END DESCRIPTION:
#Sta/Elev= 20
       0  1074.3   1.1891072.656   1.6721071.921    2.451071.228     3.5 1070.94
     7.5 1070.26     9.5 1070.16     9.8 1069.41   11.85 1069.46    13.9 1069.23
    14.9 1069.91    15.9 1070.24    16.9 1071.59    17.9  1073.7    18.9 1075.19
    19.9  1076.5    20.9 1076.84   21.05 1076.84   21.05 1076.69    25.6 1076.69
#Mann= 3 , 0 , 0
       0     .06       0     3.5    .045       0    16.9     .06       0
Levee=-1,0.05,1074.33,-1,21.03,1076.88,,
Bank Sta=3.5,16.9
XS Rating Curve= 0 ,0
Exp/Cntr=0.3,0.1

Type RM Length L Ch R = 1 ,33      ,32.067,32.167,32.233
BEGIN DESCRIPTION:
S2400
END DESCRIPTION:
#Sta/Elev= 8
       01071.577       11070.877       21069.857       31068.437       41067.827
     6.51067.727       91067.967      131068.677
#Mann= 3 , 0 , 0
       0     .06       0       2    .045       0      13     .06       0
Levee=-1,0.02,1071.6,-1,12.96,1068.69,,
Bank Sta=2,13
XS Rating Curve= 0 ,0
Exp/Cntr=0.3,0.1

Type RM Length L Ch R = 3 ,32.7    ,,,
BEGIN DESCRIPTION:
Puente Azul
END DESCRIPTION:
Bridge Culvert--1,0,-1,-1, 0
Deck Dist Width WeirC Skew NumUp NumDn MinLoCord MaxHiCord MaxSubmerge Is_Ogee
15,6,1.4,0, 6, 6, , , 0.98, 0, 0,0,,
       0      .2      .2    12.8    12.8      13
 1070.85 1070.85 1070.85 1070.85 1070.85 1070.85
    1065    1065 1070.22 1070.22    1065    1065
       0      .2      .2    12.8    12.8      13
 1070.85 1070.85 1070.85 1070.85 1070.85 1070.85
    1065    1065 1070.22 1070.22    1065    1065
BR Coef=-1 , 0 , 0 ,, 0 ,,,0.8,-1,,0,
WSPro=,,,, 1 ,,,, 0 ,,,, 0 ,,,,-1 ,-1 ,-1 , 0 , 0 , 0 , 0 , 0
BC Design=,, 0 ,, 0 ,,,,,,
BC Use User HTab Curves=0
BC User HTab FreeFlow(D)= 0

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
Type RM Length L Ch R = 1 ,32      ,33,33,33
BEGIN DESCRIPTION:
2500
END DESCRIPTION:
#Sta/Elev= 8
       01071.577       11070.877       21069.857       31068.437       4  1064.2
     6.5  1064.2       91067.967      131068.677
#Mann= 3 , 0 , 0
       0     .06       0       2    .045       0       9     .06       0
Levee=-1,0.04,1071.61,-1,12.99,1068.7,,
Bank Sta=2,9
XS Rating Curve= 0 ,0
Exp/Cntr=0.3,0.1

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
Type RM Length L Ch R = 1 ,31      ,33.263,33.267,33.28
BEGIN DESCRIPTION:
S2600
END DESCRIPTION:
#Sta/Elev= 12
       01066.948     6.31067.068     7.81066.408     8.81065.928    10.81065.048
    11.31063.678    11.81063.528   14.151063.278    16.51063.648    18.51065.268
    20.51066.568    25.51066.468
#Mann= 3 , 0 , 0
       0     .06       0    10.8    .045       0    18.5     .06       0
Levee=-1,6.37,1067.08,-1,20.55,1066.58,,
Bank Sta=10.8,18.5
XS Rating Curve= 0 ,0
Exp/Cntr=0.3,0.1

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
Type RM Length L Ch R = 3 ,30.1    ,,,
BEGIN DESCRIPTION:
PEatonal
END DESCRIPTION:
Bridge Culvert--1,0,-1,-1, 0
Deck Dist Width WeirC Skew NumUp NumDn MinLoCord MaxHiCord MaxSubmerge Is_Ogee
5,2,1.4,0, 6, 6, , , 0.98, 0, 0,0,,
       0      17      17      30      30   30.87
 1064.81 1064.81 1064.81 1064.17 1064.17 1064.17
    1060    1060 1064.66    1064    1064    1060
       0      20      20      33      33   33.49
 1064.81 1064.81 1064.81 1064.17 1064.17 1064.17
    1060    1060 1064.66    1064    1064    1060
BR Coef=-1 , 0 , 0 ,, 0 ,,,0.8,-1,,0,
WSPro=,,,, 1 ,,,, 0 ,,,, 0 ,,,,-1 ,-1 ,-1 , 0 , 0 , 0 , 0 , 0
BC Design=,, 0 ,, 0 ,,,,,,
BC Use User HTab Curves=0
BC User HTab FreeFlow(D)= 0

Type RM Length L Ch R = 1 ,30      ,99.18,99.4,99.68
BEGIN DESCRIPTION:
S2700
END DESCRIPTION:
#Sta/Elev= 13
   -.391 1064.73   5.609 1064.73   5.759 1064.84   5.759 1064.73  15.759 1064.67
  19.659 1064.56  21.159 1063.62  22.659 1062.46  25.159 1061.36  27.6091061.062
  30.059 1061.18  31.559 1064.58  33.559 1065.24
#Mann= 3 , 0 , 0
   -.391     .06       0  21.159    .045       0  31.559     .06       0
Levee=-1,5.75,1064.84,-1,33.49,1065.23,,
Bank Sta=21.159,31.559
XS Rating Curve= 0 ,0
Exp/Cntr=0.3,0.1

Type RM Length L Ch R = 1 ,29      ,96.62,99.5,103.15
BEGIN DESCRIPTION:
S2800
END DESCRIPTION:
#Sta/Elev= 11
       0 1062.22     4.2 1062.22     5.2 1061.93     6.2 1060.75     7.2 1059.96
     8.2 1059.64     9.2    1059    10.2 1058.95   12.15 1058.45    14.1 1058.55
   17.55 1063.69
#Mann= 3 , 0 , 0
       0     .06       0     4.2    .045       0   17.55     .06       0
Levee=-1,4.19,1062.25,-1,17.53,1063.71,,
Bank Sta=4.2,17.55
XS Rating Curve= 0 ,0
Exp/Cntr=0.3,0.1

Type RM Length L Ch R = 1 ,28      ,34.297,34.367,34.517
BEGIN DESCRIPTION:
S2900
END DESCRIPTION:
#Sta/Elev= 15
    -.15 1061.03       0 1061.03     3.8 1060.41     5.8 1060.13     7.8 1059.09
     8.8 1058.33     9.8 1057.57    12.2  1057.3    14.6 1057.19      161060.209
      18 1060.79      20 1060.97      22 1060.99      24 1061.09      27 1061.09
#Mann= 3 , 0 , 0
    -.15     .06       0     7.8    .045       0      16     .06       0
Levee=-1,-0.11,1061.03,-1,26.97,1061.1,,
Bank Sta=7.8,16
XS Rating Curve= 0 ,0
Exp/Cntr=0.3,0.1

Type RM Length L Ch R = 3 ,27.9    ,,,
BEGIN DESCRIPTION:
Ntra Señora
END DESCRIPTION:
Bridge Culvert--1,0,-1,-1, 0
Deck Dist Width WeirC Skew NumUp NumDn MinLoCord MaxHiCord MaxSubmerge Is_Ogee
5,6,1.4,0, 6, 6, , , 0.98, 0, 0,0,,
       0       6       6   16.15   16.15   26.97
 1060.03 1060.03 1060.03 1060.03 1060.03 1060.03
    1056    1056 1059.03 1059.03    1056    1056
       0      11      11   21.15   21.15   28.06
 1060.03 1060.03 1060.03 1060.03 1060.03 1060.03
    1056    1056 1059.03 1059.03    1056    1056
BR Coef=-1 , 0 , 0 ,, 0 ,,,0.8,-1,,0,
WSPro=,,,, 1 ,,,, 0 ,,,, 0 ,,,,-1 ,-1 ,-1 , 0 , 0 , 0 , 0 , 0
BC Design=,, 0 ,, 0 ,,,,,,
BC Use User HTab Curves=0
BC User HTab FreeFlow(D)= 0

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
Type RM Length L Ch R = 1 ,27      ,105,102.3,98.81
BEGIN DESCRIPTION:
S3000
END DESCRIPTION:
#Sta/Elev= 18
   -2.65 1063.53       0 1063.53      .5 1063.29     1.5  1063.5     8.3 1063.34
     9.9 1063.47      12 1063.08   13.25  1062.5   14.25 1061.73   15.25 1060.91
   16.25 1060.35   17.25 1059.86   18.25 1058.43   19.25 1057.53   24.25 1055.45
   25.25 1056.86   28.25 1057.36   30.25 1057.43
#Mann= 3 , 0 , 0
   -2.65     .06       0   18.25    .045       0   30.25     .06       0
Levee=-1,-0.09,1063.54,-1,30.24,1057.43,,
Bank Sta=18.25,30.25
XS Rating Curve= 0 ,0
Exp/Cntr=0.3,0.1

Type RM Length L Ch R = 1 ,26      ,97.64,98.1,99.22
BEGIN DESCRIPTION:
S3100
END DESCRIPTION:
#Sta/Elev= 14
       0 1060.36       7 1059.59     8.5 1058.84    10.5 1057.93    12.5 1057.16
    14.5 1056.85    19.5 1056.43    21.5 1055.51    23.5 1054.83    24.5 1054.77
    29.5 1053.06      33 1054.96   36.65 1055.36    36.8 1055.36
#Mann= 3 , 0 , 0
       0     .06       0    19.5    .045       0   36.65     .06       0
Levee=-1,0.19,1060.38,-1,36.69,1055.41,,
Bank Sta=19.5,36.65
XS Rating Curve= 0 ,0
Exp/Cntr=0.3,0.1

Type RM Length L Ch R = 1 ,25      ,98.71,99.1,100.64
BEGIN DESCRIPTION:
S3200
END DESCRIPTION:
#Sta/Elev= 11
       0 1053.18       1 1051.74       2 1051.76    2.97 1051.23     5.5 1050.92
    8.03 1051.08    9.03 1052.03   11.03 1053.53   12.03  1054.4   16.53 1054.28
   24.03 1054.19
#Mann= 3 , 0 , 0
       0     .06       0       2    .045       0    9.03     .06       0
Levee=-1,0.04,1053.18,-1,12.03,1054.41,,
Bank Sta=2,9.03
XS Rating Curve= 0 ,0
Exp/Cntr=0.3,0.1

Type RM Length L Ch R = 1 ,24      ,99.28,96.5,93.3
BEGIN DESCRIPTION:
S3300
END DESCRIPTION:
#Sta/Elev= 10
       0 1053.92     2.2  1053.5     4.4 1052.96     7.4 1052.24    10.4    1050
    11.9 1048.98    14.4 1048.96    16.9 1048.96    18.9 1049.59    20.9 1049.85
#Mann= 3 , 0 , 0
       0     .06       0    10.4    .045       0    18.9     .06       0
Levee=-1,0.06,1053.92,-1,20.89,1049.86,,
Bank Sta=10.4,18.9
XS Rating Curve= 0 ,0
Exp/Cntr=0.3,0.1

Type RM Length L Ch R = 1 ,23      ,97.05,99.5,101.94
BEGIN DESCRIPTION:
S3400
END DESCRIPTION:
#Sta/Elev= 12
       0  1049.9       5  1049.9       6  1048.6      10 1048.38      15 1047.55
    15.5 1047.31    18.5 1047.34    21.5 1047.48    22.3  1048.8    24.3 1048.83
    26.3 1049.01    31.3 1049.01
#Mann= 3 , 0 , 0
       0     .06       0       6    .045       0    22.3     .06       0
Levee=-1,4.97,1049.9,-1,26.27,1049.01,,
Bank Sta=6,22.3
XS Rating Curve= 0 ,0
Exp/Cntr=0.3,0.1

Type RM Length L Ch R = 1 ,22      ,100.6,101.8,103.15
BEGIN DESCRIPTION:
S3500
END DESCRIPTION:
#Sta/Elev= 10
       0 1048.78    10.3 1048.76    12.3 1048.12    13.9 1046.61    14.9 1045.74
   17.45 1045.49      20 1045.66      21  1046.3      22 1046.61      24 1046.84
#Mann= 3 , 0 , 0
       0     .06       0    12.3    .045       0      24     .06       0
Levee=-1,10.31,1048.77,-1,24,1046.85,,
Bank Sta=12.3,24
XS Rating Curve= 0 ,0
Exp/Cntr=0.3,0.1

Type RM Length L Ch R = 1 ,21      ,107.6,105.8,103.47
BEGIN DESCRIPTION:
S3600
END DESCRIPTION:
#Sta/Elev= 12
       0  1044.8     9.6  1044.9    12.6  1044.1    14.6  1043.6    15.1    1043
    17.4  1042.5    19.6    1043    20.1  1043.2    21.6  1043.2    23.7  1043.6
    25.4  1044.5    25.5  1044.5
#Mann= 3 , 0 , 0
       0     .06       0    14.6    .045       0    23.7     .06       0
Levee=-1,9.59,1044.91,-1,25.53,1044.5,,
Bank Sta=14.6,23.7
XS Rating Curve= 0 ,0
Exp/Cntr=0.3,0.1

Type RM Length L Ch R = 1 ,20      ,99.25,98.6,97.6
BEGIN DESCRIPTION:
S3700
END DESCRIPTION:
#Sta/Elev= 15
       0 1041.79       1 1041.79       2 1041.31       4 1040.78       6 1040.32
     6.5 1039.89     9.2 1039.74    11.9 1040.01    12.9 1040.81    13.9 1041.32
    14.9 1042.01    16.4 1044.31    17.7 1044.31   17.85 1044.31  19.288 1044.31
#Mann= 3 , 0 , 0
       0     .06       0       2    .045       0    14.9     .06       0
Levee=-1,0.97,1041.79,-1,16.4,1044.31,,
Bank Sta=2,14.9
XS Rating Curve= 0 ,0
Exp/Cntr=0.3,0.1

Type RM Length L Ch R = 1 ,19      ,116.8,104.2,112.03
BEGIN DESCRIPTION:
S3800
END DESCRIPTION:
#Sta/Elev= 12
       0 1040.63       8 1040.24       9 1040.29    10.8 1039.46    11.8 1038.54
    14.3 1038.39    16.8 1038.39    18.3 1039.39    20.3 1040.52    22.3 1042.42
    23.3 1042.56   23.45 1042.56
#Mann= 3 , 0 , 0
       0     .06       0       9    .045       0    20.3     .06       0
Levee=-1,0.08,1040.65,-1,23.36,1042.57,,
Bank Sta=9,20.3
XS Rating Curve= 0 ,0
Exp/Cntr=0.3,0.1

Type RM Length L Ch R = 1 ,18      ,96.58,96.5,96.44
BEGIN DESCRIPTION:
S3900
END DESCRIPTION:
#Sta/Elev= 17
      .3 1041.85      .3  1039.4     1.3  1039.4     1.3  1038.4     3.1 1038.18
     3.2 1037.15     4.2  1037.2     6.2 1037.37     8.2 1037.54    10.2 1036.77
    12.2 1036.76    14.2 1036.85    16.2 1037.13    18.2 1037.57    20.2  1038.4
    20.2  1041.9    20.7  1041.9
#Mann= 3 , 0 , 0
      .3     .06       0     3.1    .045       0    18.2     .06       0
Levee=-1,0.29,1041.88,-1,20.15,1041.91,,
Bank Sta=3.1,18.2
XS Rating Curve= 0 ,0
Exp/Cntr=0.3,0.1

Type RM Length L Ch R = 1 ,17      ,101.4,100.5,99.5
BEGIN DESCRIPTION:
S4000
END DESCRIPTION:
#Sta/Elev= 11
       0 1036.94       2 1035.83       5 1034.83     5.5 1034.35    8.051034.242
    10.6 1034.26    11.6 1035.74    13.6 1035.94    14.6 1037.16    17.8 1041.16
  20.3721041.168
#Mann= 3 , 0 , 0
       0     .06       0       2    .045       0    11.6     .06       0
Levee=-1,0.02,1036.99,-1,17.84,1041.22,,
Bank Sta=2,11.6
XS Rating Curve= 0 ,0
Exp/Cntr=0.3,0.1

Type RM Length L Ch R = 1 ,16      ,92.43,95.2,99.14
BEGIN DESCRIPTION:
S4100
END DESCRIPTION:
#Sta/Elev= 11
       0 1035.56    4.24 1035.56    5.24 1034.37    6.24 1033.71    7.24 1032.36
   10.54 1032.32   13.84 1032.33   14.84 1033.18   15.84 1033.51   16.84 1034.31
   17.84 1035.49
#Mann= 3 , 0 , 0
       0     .06       0    6.24    .045       0   16.84     .06       0
Levee=-1,4.26,1035.56,-1,17.79,1035.49,,
Bank Sta=6.24,16.84
XS Rating Curve= 0 ,0
Exp/Cntr=0.3,0.1

Type RM Length L Ch R = 1 ,15      ,35.27,34.4,33.963
BEGIN DESCRIPTION:
S4200
S4200
END DESCRIPTION:
#Sta/Elev= 12
       01035.838     2.81030.768     5.61030.989     9.61031.747    13.11033.277
    17.61035.137    25.11035.587    29.61035.508   32.451035.048   32.451035.508
    32.61035.048    39.41035.048
#Mann= 3 , 0 , 0
       0     .06       0       0    .045       0    13.1     .06       0
Levee=-1,0.06,1035.86,-1,25.11,1035.61,,
Bank Sta=0,13.1
XS Rating Curve= 0 ,0
Exp/Cntr=0.3,0.1

Type RM Length L Ch R = 3 ,14.8    ,,,
BEGIN DESCRIPTION:
Puente Bomberos
END DESCRIPTION:
Bridge Culvert--1,0,-1,-1, 0
Deck Dist Width WeirC Skew NumUp NumDn MinLoCord MaxHiCord MaxSubmerge Is_Ogee
5,6,1.4,0, 6, 6, , , 0.98, 0, 0,0,,
       0       1       1    11.8    11.8    39.4
 1033.85 1033.85 1033.85 1033.85 1033.85 1033.85
    1030    1030 1032.85 1032.85    1030    1030
       0       6       6    16.8    16.8   38.87
 1033.85 1033.85 1033.85 1033.85 1033.85 1033.85
    1030    1030 1032.85 1032.85    1030    1030
BR Coef=-1 , 0 , 0 ,, 0 ,,,0.8,-1,,0,
WSPro=,,,, 1 ,,,, 0 ,,,, 0 ,,,,-1 ,-1 ,-1 , 0 , 0 , 0 , 0 , 0
BC Design=,, 0 ,, 0 ,,,,,,
BC Use User HTab Curves=0
BC User HTab FreeFlow(D)= 0

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
Type RM Length L Ch R = 1 ,14      ,107.5,107.05,107.05
BEGIN DESCRIPTION:
S4300
END DESCRIPTION:
#Sta/Elev= 13
       0  1032.8    10.6  1032.8    12.2  1030.2    14.5  1029.8    16.1  1029.3
    19.6    1029    23.1  1029.1      24    1030      24  1029.1    27.5  1030.5
    32.4  1032.8    36.5  1034.2    37.8  1034.2
#Mann= 3 , 0 , 0
       0     .06       0    12.2    .045       0    27.5     .06       0
Levee=-1,10.56,1032.83,-1,36.57,1034.22,,
Bank Sta=12.2,27.5
XS Rating Curve= 0 ,0
Exp/Cntr=0.3,0.1

Type RM Length L Ch R = 1 ,13      ,93.38,95.3,98.8
BEGIN DESCRIPTION:
S4400
END DESCRIPTION:
#Sta/Elev= 12
       0 1028.68     3.9 1028.97     7.9 1028.32     8.4 1027.73    10.9 1027.64
    13.4  1027.8    20.9 1027.99    24.9 1028.78    26.1 1031.17    33.1 1033.77
    45.9 1033.77  48.301 1033.77
#Mann= 3 , 0 , 0
       0     .06       0     3.9    .045       0    24.9     .06       0
Levee=-1,3.82,1028.99,-1,33.17,1033.79,,
Bank Sta=3.9,24.9
XS Rating Curve= 0 ,0
Exp/Cntr=0.3,0.1

Type RM Length L Ch R = 1 ,12      ,98.76,99.1,99.63
BEGIN DESCRIPTION:
S4500
END DESCRIPTION:
#Sta/Elev= 19
    -.151029.845       0 1027.84       01029.845    3.76 1025.39    7.73 1025.26
   11.73 1025.24   12.88 1026.14   17.88 1026.26   20.58 1028.31   22.88 1029.54
   25.57 1031.13   25.57 1030.84  26.363 1031.13   30.57 1032.64   33.07 1032.64
  35.0431032.389  35.4771031.862   35.57 1031.14   38.57 1031.14
#Mann= 3 , 0 , 0
    -.15     .06       0       0    .045       0   17.88     .06       0
Levee=-1,0.04,1029.86,-1,30.62,1032.67,,
Bank Sta=0,17.88
XS Rating Curve= 0 ,0
Exp/Cntr=0.3,0.1

Type RM Length L Ch R = 1 ,11      ,107.91,104.2,96.66
BEGIN DESCRIPTION:
S4600
END DESCRIPTION:
#Sta/Elev= 20
    -.03 1030.85    -.03 1029.03    9.97 1026.03   20.17 1025.26   21.57 1024.12
   25.07 1024.13   28.57 1024.22   29.17 1024.22   29.17 1024.83   34.17 1025.27
   36.77 1027.36   40.57 1028.65   43.57 1032.06   46.97 1032.26   51.97 1028.44
   55.77 1028.44   55.77 1030.44   55.92 1030.44   55.92 1028.44   58.64 1028.44
#Mann= 3 , 0 , 0
    -.03     .06       0    9.97    .045       0   34.17     .06       0
Levee=-1,-0.11,1030.87,-1,46.97,1032.26,,
Bank Sta=9.97,34.17
XS Rating Curve= 0 ,0
Exp/Cntr=0.3,0.1

Type RM Length L Ch R = 1 ,10      ,104.3,102.8,101.55
BEGIN DESCRIPTION:
S4700
END DESCRIPTION:
#Sta/Elev= 29
   -3.11 1039.97    -2.4 1039.58   -1.94 1038.94   -1.09 1038.58       0 1037.53
     .34 1036.49    1.02 1034.29    1.59 1032.45    2.64 1029.79    3.24 1028.46
    3.88 1026.87     5.3  1024.7     9.3 1024.23    10.3 1023.42    15.3 1023.52
    20.3 1023.14    22.8 1022.97    25.3 1022.85    26.8 1023.78    27.8 1024.79
    28.8 1025.25    33.8 1028.61    36.3  1031.1   37.52 1032.58    41.3 1032.58
   42.63  1030.4   43.48    1029   44.26 1028.26    46.3 1027.84
#Mann= 3 , 0 , 0
   -3.11     .06       0     5.3    .045       0    27.8     .06       0
Levee=-1,-2.77,1039.91,-1,37.58,1032.65,,
Bank Sta=5.3,27.8
XS Rating Curve= 0 ,0
Exp/Cntr=0.3,0.1

Type RM Length L Ch R = 1 ,9       ,102.56,100.5,99.53
BEGIN DESCRIPTION:
S4800
END DESCRIPTION:
#Sta/Elev= 28
       0  1027.2       1  1022.5       2  1022.4       3  1022.3     3.5  1022.3
       4  1022.3       5  1022.3       6  1022.3       7  1022.5       8  1022.6
       9  1022.7      10  1022.9      11    1023      12  1023.8      13  1024.7
      14  1025.6      15  1026.6      16  1027.5      17  1028.4      18  1029.2
      19  1030.3      20  1030.3      21  1030.2      22  1030.3      23  1030.2
      24  1030.2      25  1030.2      26  1030.2
#Mann= 3 , 0 , 0
       0     .06       0       0    .045       0      12     .06       0
Levee=-1,0.05,1027.27,-1,19.02,1030.34,,
Bank Sta=0,12
XS Rating Curve= 0 ,0
Exp/Cntr=0.3,0.1

Type RM Length L Ch R = 1 ,8       ,93.7,95.2,97.16
BEGIN DESCRIPTION:
S4900
END DESCRIPTION:
#Sta/Elev= 17
       0  1023.5     2.7  1023.5     2.9  1023.5     5.2  1023.5     7.6  1023.5
     7.6  1023.8    10.3  1023.8    10.6  1023.8    10.6  1021.3    15.3  1020.5
    19.8  1020.5    23.8  1023.7    25.1  1025.2    25.8  1026.8    26.2  1027.9
    26.6  1029.5    28.6  1029.5
#Mann= 3 , 0 , 0
       0     .06       0    10.6    .045       0    23.8     .06       0
Levee=-1,7.64,1023.84,-1,26.59,1029.49,,
Bank Sta=10.6,23.8
XS Rating Curve= 0 ,0
Exp/Cntr=0.3,0.1

Type RM Length L Ch R = 1 ,7       ,97.23,96.7,96.15
BEGIN DESCRIPTION:
S5000
END DESCRIPTION:
#Sta/Elev= 14
       0  1027.2     2.2  1027.2     2.2  1019.2    12.2  1019.3    14.7    1020
    17.7  1020.8    21.7  1022.6    22.8  1023.1    28.8  1023.1      32  1023.2
   32.19 1018.59    32.2  1018.4    32.2  1018.3    38.6  1018.3
#Mann= 3 , 0 , 0
       0     .06       0     2.2    .045       0    17.7     .06       0
Levee=-1,2.07,1027.22,-1,31.91,1023.27,,
Bank Sta=2.2,17.7
XS Rating Curve= 0 ,0
Exp/Cntr=0.3,0.1

Type RM Length L Ch R = 1 ,6       ,98.6,99.8,100.67
BEGIN DESCRIPTION:
S5100
END DESCRIPTION:
#Sta/Elev= 11
       0  1023.5       3 1023.34     6.5 1023.62       9 1022.04     9.9 1020.84
    11.9 1020.77    14.1 1018.43    17.1 1018.53    20.1 1018.65    26.1    1019
    33.1 1022.85
#Mann= 3 , 0 , 0
       0     .06       0    11.9    .045       0    33.1     .06       0
Levee=-1,6.54,1023.6,-1,33.03,1022.86,,
Bank Sta=11.9,33.1
XS Rating Curve= 0 ,0
Exp/Cntr=0.3,0.1

Type RM Length L Ch R = 1 ,5       ,114.36,110.1,106.32
BEGIN DESCRIPTION:
S5200
END DESCRIPTION:
#Sta/Elev= 13
       0 1018.19     2.9 1018.19     6.5 1019.29     8.6 1019.34     8.9 1019.34
     8.9 1017.57    15.4 1016.82    21.9 1016.39    22.4 1017.39    23.6 1017.86
    23.9 1018.86    31.9 1021.22    31.9 1023.22
#Mann= 3 , 0 , 0
       0     .06       0     8.9    .045       0    23.6     .06       0
Levee=-1,8.62,1019.34,-1,31.92,1023.23,,
Bank Sta=8.9,23.6
XS Rating Curve= 0 ,0
Exp/Cntr=0.3,0.1

Type RM Length L Ch R = 1 ,4       ,99.67,99.78,99.96
BEGIN DESCRIPTION:
S5300
END DESCRIPTION:
#Sta/Elev= 16
       0 1021.34       6 1021.34       6  1021.6     7.5  1021.6     7.5 1021.85
     9.6 1021.85   12.65 1018.83    15.3 1017.64    18.2  1015.5    23.4 1015.15
    28.6 1015.47    29.1 1015.87    33.1 1018.26    37.1 1020.07    40.1 1019.97
    40.1 1021.97
#Mann= 3 , 0 , 0
       0     .06       0    15.3    .045       0    33.1     .06       0
Levee=-1,9.61,1021.88,-1,40.08,1021.99,,
Bank Sta=15.3,33.1
XS Rating Curve= 0 ,0
Exp/Cntr=0.3,0.1

Type RM Length L Ch R = 1 ,3       ,98.3,100.2,101.13
BEGIN DESCRIPTION:
S5400
END DESCRIPTION:
#Sta/Elev= 17
       0  1018.5       6  1018.6      16  1019.1      26  1019.3      36  1019.6
      53  1019.5      54  1017.5    55.9  1016.3      57  1015.2    60.2    1014
      62  1013.8    65.8  1013.4    69.5  1013.8    72.2  1014.1    75.1  1014.9
    77.6  1018.7    80.6  1019.4
#Mann= 3 , 0 , 0
       0     .06       0      57    .045       0    75.1     .06       0
Levee=-1,36.22,1019.62,-1,80.54,1019.39,,
Bank Sta=57,75.1
XS Rating Curve= 0 ,0
Exp/Cntr=0.3,0.1

Type RM Length L Ch R = 1 ,2       ,96.77,97.2,98.44
BEGIN DESCRIPTION:
S5500
END DESCRIPTION:
#Sta/Elev= 15
       0 1018.31     7.4 1018.08   9.685 1017.35    11.2 1015.92    11.2 1015.52
      15 1012.14   19.25 1012.14    23.5 1012.22    23.9 1012.42    26.7 1012.67
    28.5 1014.08    32.9 1017.45    35.9 1017.37    40.9 1017.32    46.9 1017.19
#Mann= 3 , 0 , 0
       0     .06       0    11.2    .045       0    28.5     .06       0
Levee=-1,0.12,1018.35,-1,33.01,1017.48,,
Bank Sta=11.2,28.5
XS Rating Curve= 0 ,0
Exp/Cntr=0.3,0.1

Type RM Length L Ch R = 1 ,1       ,0,0,0
BEGIN DESCRIPTION:
S5600
END DESCRIPTION:
#Sta/Elev= 21
       0 1014.66    1.46 1014.66    1.46 1014.95    8.66 1014.98    8.66 1014.62
   12.86 1014.72   21.86  1014.5   26.86 1014.17   31.86 1013.61   37.86 1012.83
   38.18 1012.83   38.18 1012.21   40.58 1011.48   41.58 1010.69   42.98  1011.1
   43.38 1010.69   46.25 1010.89   49.44 1011.19   49.44 1012.39   49.74 1012.39
   49.74 1016.23
#Mann= 3 , 0 , 0
       0     .06       0   38.18    .045       0   49.44     .06       0
Levee=-1,8.69,1014.95,-1,49.69,1016.21,,
Bank Sta=38.18,49.44
XS Rating Curve= 0 ,0
Exp/Cntr=0.3,0.1

Chan Stop Cuts=-1
Use User Specified Reach Order=0
